HEC-RAS study BRSHRN.prj: BRSHRN

--- BRSHRN.g01 (geometry) --- (continued)

Type RM Length L Ch R = 1 ,16733   ,472.4,495.1,505.3
XS GIS Cut Line= 4
2310269.19010119551055.432507611 2310250.7414884551150.368133767
2310317.66051564 551501.728842492310517.28573329551672.325791578
#Sta/Elev= 30
       0 2801.15    18.1 2795.49    34.4 2792.14    50.7 2791.09    71.1 2788.12
    96.7 2786.29   134.5 2779.99   156.6 2778.56   165.62776.766   172.9 2775.59
   180.92776.683   189.2 2777.56   201.4 2777.31   224.2 2778.34   270.6 2777.64
   315.8 2778.28   363.7 2780.13   388.7 2780.25   425.3 2782.38   475.6 2782.38
   515.4  2782.9   533.6 2783.79   545.9 2783.47   562.9 2784.08   583.5 2784.05
   615.5  2784.9   626.1 2785.72     643 2786.12   694.5 2788.65     717 2788.52
#Mann= 8 ,-1,0
       0     .12       0      50      .1       0  146.71     .08       0
   165.6    .045       0   180.9     .08       0  446.71     .07       0
  594.39     .06       0  674.39      .1       0
Bank Sta=165.6,180.9
XS Rating Curve= 0 ,0
Exp/Cntr(USF)=0,0
Exp/Cntr=0.3,0.1

Type RM Length L Ch R = 1 ,16238   ,419.4,417.5,410.8
XS GIS Cut Line= 3
2310189.33273144551038.9505362482310130.89972533551247.343632063
 2309870.2614159551499.443114394
#Sta/Elev= 30
       0 2796.28    10.6    2794    19.1 2792.79    68.8 2787.67    89.6 2787.77
     102 2786.46   114.5 2786.53   122.8 2785.97   147.7  2780.4   164.3 2779.44
   176.8 2778.04     210 2776.63   219.1 2777.13   236.3 2776.57   259.3 2777.12
   270.3  2775.7   281.4 2775.23     296 2776.26   314.8 2775.88   355.4 2776.72
   361.1 2776.13   364.9  2774.5   372.4 2773.56   378.1 2773.67   383.92774.635
   392.2 2775.27   406.4 2774.28     415 2777.06   491.2 2781.23     579 2782.13
#Mann= 6 ,-1,0
       0     .12       0      20      .1       0  286.43     .08       0
   364.9    .045       0   383.9     .08       0  416.43     .05       0
Bank Sta=364.9,383.9
XS Rating Curve= 0 ,0
Exp/Cntr(USF)=0,0
Exp/Cntr=0.3,0.1

Type RM Length L Ch R = 1 ,15820   ,410.7,409.1,403.9
XS GIS Cut Line= 3
2309903.46977981550957.1541236792309697.75425119 551358.78920336
2309686.32561071 551438.78968671
#Sta/Elev= 30
       0 2794.49    24.8 2793.41      54 2791.51    58.5 2790.89    62.9 2789.38
    89.9 2775.81    94.4 2774.22    98.9 2774.15   118.4 2775.35   130.1 2775.03
   157.3 2775.32   192.7 2774.26   211.3 2774.77   251.7 2775.05   269.9 2774.19
   278.1 2772.26   281.8 2771.61   287.8 2771.31   292.1 2771.34   295.4 2772.21
   296.7 2772.61   301.1 2775.09   305.6 2775.34   319.1 2774.77   337.1 2775.76
     367 2776.57   418.5 2779.31   457.7 2779.07   498.1 2781.45   532.1 2781.53
#Mann= 8 ,-1,0
       0     .12       0      30      .1       0      50     .12       0
     270     .05       0   278.1    .045       0   295.4     .05       0
     380     .08       0  481.25     .05       0
Bank Sta=278.1,295.4
XS Rating Curve= 0 ,0
Exp/Cntr(USF)=0,0
Exp/Cntr=0.3,0.1

Type RM Length L Ch R = 1 ,15411   ,261.4,258.3,254.6
XS GIS Cut Line= 2
2309593.26382395550904.908910062 2309487.1407338551428.993709157
#Sta/Elev= 30
       0 2791.88    20.7 2789.41    28.8 2788.88    48.7  2786.5    62.2 2785.16
    77.8 2784.11   102.3  2783.8   106.4 2783.16   110.5 2781.76   122.7 2776.06
   136.9 2772.43   143.1 2770.73   146.6 2770.62   147.4 2770.69   152.5 2772.32
   155.4 2773.28   159.4 2773.62   167.6 2773.25   179.8 2773.69   228.8 2773.47
   269.6 2774.22   326.8 2774.28     339 2774.87   359.4 2776.52   400.2 2778.04
   424.7 2778.39   452.5 2779.53   500.1 2780.75   522.7 2781.86   534.7 2782.76
#Mann= 4 ,-1,0
       0      .1       0   136.9    .045       0   152.5      .1       0
     200     .05       0
Bank Sta=136.9,152.5
XS Rating Curve= 0 ,0
Exp/Cntr(USF)=0,0
Exp/Cntr=0.3,0.1

Type RM Length L Ch R = 1 ,15153   ,451.9,459.4,458
XS GIS Cut Line= 2
2309313.15687154550885.0614526672309333.23195419551417.051142933
#Sta/Elev= 30
       0 2793.24    12.1 2789.51    28.1 2785.19    45.5 2781.18    52.2 2779.96
    76.2 2777.44    80.2 2776.25    84.3 2774.25    91.7 2772.02    96.2 2771.33
   100.2 2771.37   103.3  2770.6   108.2 2769.66   112.2 2769.62   122.6 2770.42
   140.2 2772.28   156.2 2773.47   164.2 2772.96   176.2 2772.68   252.3 2773.73
   284.3 2773.15   321.4 2773.25   336.4 2773.85   356.4 2775.31   392.2 2776.67
   416.4 2778.31   440.4 2778.68   464.4 2779.87   500.5 2780.87   532.4 2782.24
#Mann= 6 ,-1,0
       0     .12       0      20      .1       0   103.3    .045       0
   122.6      .1       0     220     .07       0     310     .05       0
Bank Sta=103.3,122.6
XS Rating Curve= 0 ,0
Exp/Cntr(USF)=0,0
Exp/Cntr=0.3,0.1

Type RM Length L Ch R = 1 ,14693   ,464.3,469.6,467.3
XS GIS Cut Line= 3
 2308936.2211034550885.2871584862309032.01356584551393.312532959
2309162.24081161551481.238922774
#Sta/Elev= 30
       0 2790.29    12.1 2787.44    20.4 2786.18    36.5 2786.67    48.7 2786.23
      65 2785.15    85.4 2782.73    97.6  2780.3   109.8 2773.87   113.9  2773.2
   191.7 2772.91   223.8 2771.99     240  2773.3   256.3 2773.47   264.5 2773.23
   280.7 2771.59   313.3 2772.47   317.4 2771.77   323.6 2769.75     326 2769.14
   337.7 2769.39   349.2  2768.8   357.42769.717   362.9  2771.5   370.3 2772.71
   402.9 2774.92   500.6 2778.06   559.6 2777.95   623.6 2782.56   674.1 2782.99
#Mann= 6 ,-1,0
       0      .1       0   323.6    .045       0   357.4      .1       0
     420     .05       0  516.98     .08       0  606.98     .05       0
Bank Sta=323.6,357.4
XS Rating Curve= 0 ,0
Exp/Cntr(USF)=0,0
Exp/Cntr=0.3,0.1

Type RM Length L Ch R = 1 ,14224   ,449.9,453.8,444.1
XS GIS Cut Line= 2
2308612.03340571551048.583247509 2308726.3198105551541.647451019
#Sta/Elev= 30
       0 2785.68    25.2 2782.72    33.5 2779.71    45.8 2773.59    53.9 2771.69
   100.6 2771.89   123.8 2770.45   127.3 2768.84     132 2767.11     144 2766.94
   148.4 2767.26     154 2768.64   160.7 2769.75   173.1 2769.66   181.3 2770.68
   230.6 2769.93     247 2770.92   260.6 2770.89   279.8 2770.26     284  2770.5
   296.2 2773.53   300.4 2773.81   316.8 2773.36   333.2 2774.22     366    2774
   407.3 2775.28   435.9 2775.38   457.3  2777.4   485.1 2784.13   506.1 2786.69
#Mann= 5 ,-1,0
       0      .1       0   127.3    .045       0     154      .1       0
     260     .08       0     360     .05       0
#XS Ineff= 2 , 0
                          333.33         2781.44
Permanent Ineff=
       F       F
Bank Sta=127.3,154
XS Rating Curve= 0 ,0
Exp/Cntr(USF)=0,0
Exp/Cntr=0.3,0.1

Type RM Length L Ch R = 1 ,13770   ,269.4,262.3,258.8
XS GIS Cut Line= 2
2308378.56260736551193.8902478812308533.66558529551585.729350008
#Sta/Elev= 30
       0 2789.75    16.4 2786.01    29.3 2781.27    37.7  2778.9    50.9 2777.46
    59.5 2775.59    63.8 2774.13    68.1 2771.84    71.6 2769.31    74.2 2767.89
    76.7 2766.57      81 2765.91    85.3 2765.84    99.3 2765.92   102.5 2766.21
   108.6 2767.74   128.3 2769.26   145.5  2768.5   166.8 2769.96   214.3 2769.77
   227.2 2770.77   234.9 2771.87   248.7 2772.61   284.2 2771.69   304.7  2772.4
   326.2 2773.77   347.7 2774.36   369.2 2776.16   386.4 2779.73   421.4 2782.43
#Mann= 4 ,-1,0
       0      .1       0    74.2    .045       0   108.6      .1       0
     320     .05       0
Bank Sta=74.2,108.6
XS Rating Curve= 0 ,0
Exp/Cntr(USF)=0,0
Exp/Cntr=0.3,0.1

Type RM Length L Ch R = 1 ,13508   ,442.7,443.5,441.7
XS GIS Cut Line= 2
2308080.88178181551223.7557863392308410.67969277551649.880809902
#Sta/Elev= 30
       0 2787.79    27.1 2782.98    66.1  2778.4    77.5 2776.45    83.8 2775.88
    96.9 2773.26   120.3 2770.88     126  2769.2   133.3 2766.18   137.4  2764.9
   148.5 2764.28   157.3 2764.42   163.7 2765.71   173.8 2765.82     183    2768
   185.8 2768.14   209.2 2768.19   244.6 2767.19   271.4 2767.32   299.5 2768.37
   332.2 2767.39   360.9 2768.93   401.4 2768.42   419.7 2768.78   433.9 2769.81
   446.9 2771.33   462.1 2775.29   473.8 2779.02   482.3 2780.53   538.8 2782.82
#Mann= 7 ,-1,0
       0      .1       0   133.3    .045       0   163.7      .1       0
     230     .08       0     340      .1       0     390     .08       0
     470      .1       0
#XS Ineff= 2 , 0
                           398.4         2778.39
Permanent Ineff=
       F       F
Bank Sta=133.3,163.7
XS Rating Curve= 0 ,0
Exp/Cntr(USF)=0,0
Exp/Cntr=0.3,0.1

Type RM Length L Ch R = 1 ,13064   ,394.9,397.3,394.4
XS GIS Cut Line= 3
2307864.14577845551369.2097263742307936.91356504551409.667113669
2308149.82913715551790.534720936
#Sta/Elev= 30
       0 2781.47    41.2 2778.37    64.1 2777.95   108.8 2775.25   128.5 2772.61
   146.9 2770.81   170.5 2767.15   178.9 2767.06   204.7 2765.82     244 2765.33
   252.3 2764.57   264.6 2764.17   274.12762.688   286.7 2762.16   288.9 2762.21
   293.5 2763.16   298.1 2764.51   302.8 2765.21   311.8 2765.73     321  2765.2
   325.6 2765.82   330.2 2767.07   334.7 2767.31   366.8 2766.45   389.7  2766.9
   409.6 2769.33   426.8 2772.19   455.7 2774.31   499.7 2780.62   519.6 2782.14
#Mann= 4 ,-1,0
       0      .1       0   274.1    .045       0   293.5     .08       0
  463.26      .1       0
Bank Sta=274.1,293.5
XS Rating Curve= 0 ,0
Exp/Cntr(USF)=0,0
Exp/Cntr=0.3,0.1

Type RM Length L Ch R = 1 ,12667   ,334.5,336.3,335.3
XS GIS Cut Line= 2
2307637.60021606551409.3465808882307963.36270443551949.229557298
#Sta/Elev= 30
       0 2800.66    33.8  2786.1    54.2 2778.58    60.5 2776.98    97.9 2773.16
   121.2 2771.78   158.6  2772.8   186.7  2771.8   191.3  2771.2   202.8 2765.72
     210 2763.42     2132762.734   223.2 2760.92   233.4  2762.8     245 2764.53
   266.1 2764.45   290.2 2765.51   304.8  2764.7   317.5 2766.52   354.9 2765.06
   376.6 2766.09     398 2765.64   427.1 2767.06   448.3 2766.48   470.9 2767.81
   569.8 2768.47   574.4 2769.41   604.9 2779.66   616.6 2781.35   630.6 2782.11
#Mann= 7 ,-1,0
       0      .1       0     210     .08       0     213    .045       0
   233.4     .08       0     370      .1       0     440     .08       0
     560      .1       0
#XS Ineff= 2 , 0
                          491.69         2782.33
Permanent Ineff=
       F       F
Bank Sta=213,233.4
XS Rating Curve= 0 ,0
Exp/Cntr(USF)=0,0
Exp/Cntr=0.3,0.1

Type RM Length L Ch R = 1 ,12330   ,325.6,327.5,327.5
XS GIS Cut Line= 2
2307407.93077716551601.4233742722307679.03445595552072.218055478
#Sta/Elev= 30
       0 2810.68    18.2 2801.93    59.7  2779.3    70.3 2774.21    78.2 2771.44
    84.9 2769.96      92 2769.08   133.6 2765.88   142.8 2765.73   152.8 2764.67
   160.8  2764.4     164 2763.05     167 2761.38   170.5 2760.32   178.7 2760.14
   184.5 2760.67     189 2762.31   193.6 2763.53   225.9 2764.88   262.8 2764.71
   281.3 2763.72   305.1 2764.53   327.4 2766.77     369 2766.53   417.3 2768.45
   442.8 2767.72   459.9 2768.11   479.8 2769.53   512.1 2776.89   543.3 2779.92
#Mann= 5 ,-1,0
       0      .1       0     100     .08       0     164    .045       0
     189     .08       0     440     .12       0
#XS Ineff= 2 , 0
                          332.17         2779.95
Permanent Ineff=
       F       F
Bank Sta=164,189
XS Rating Curve= 0 ,0
Exp/Cntr(USF)=0,0
Exp/Cntr=0.3,0.1

Type RM Length L Ch R = 1 ,12003   ,332,332.5,334.8
XS GIS Cut Line= 2
2307186.33045501551770.957484621  2307343.572044552069.693008068
#Sta/Elev= 30
       0 2805.21       7 2804.08    29.6    2798    38.7  2796.1    46.9 2793.22
    79.4 2780.52    83.9 2777.91   103.7 2761.89     107 2760.56     120 2760.01
   124.6 2760.44   127.4 2761.32   133.3 2762.85   138.1 2763.09     150 2762.82
   165.2 2760.84   175.7 2760.52   183.7 2760.76   192.5 2762.49   235.8 2763.26
   261.6  2763.2   278.2 2762.19   282.8 2763.42   287.3 2765.35   291.8 2766.44
   305.1 2767.92   313.1 2771.47   318.9 2773.46   323.4 2774.19   337.6  2775.3
#Mann= 4 ,-1,0
       0      .1       0   103.7    .045       0   127.4      .1       0
     240     .12       0
Bank Sta=103.7,127.4
XS Rating Curve= 0 ,0
Exp/Cntr(USF)=0,0
Exp/Cntr=0.3,0.1

Type RM Length L Ch R = 1 ,11670   ,214.6,218.5,222.5
XS GIS Cut Line= 2
2307004.58140141551875.1719669962307151.37412505552236.202719718
#Sta/Elev= 30
       0 2800.01      41 2782.12    49.7 2778.66    58.3 2773.73    71.3 2763.52
    75.6 2761.89    84.1 2761.54    88.5 2762.73    92.8    2763    97.2 2762.83
   105.8 2761.62   118.8 2763.15     137 2763.43     149  2764.2   179.2 2763.35
   196.5 2761.31   209.4 2759.96   219.2  2761.2   246.8 2761.83   265.6 2761.54
   269.9 2762.08   274.4  2763.3   282.8  2764.4   295.8 2765.05   304.4 2767.72
   317.4 2768.56     339 2771.88   363.5 2777.19   381.9 2780.67   389.7 2781.69
#Mann= 4 ,-1,0
       0      .1       0   196.5    .045       0   219.2      .1       0
     330     .08       0
Bank Sta=196.5,219.2
XS Rating Curve= 0 ,0
Exp/Cntr(USF)=0,0
Exp/Cntr=0.3,0.1

Type RM Length L Ch R = 1 ,11452   ,194.3,197.1,197
XS GIS Cut Line= 2
2306843.24165111551906.9109342682306900.10730081552295.713283354
#Sta/Elev= 30
       0 2805.43    10.4 2801.49    34.6 2790.43    46.8 2785.94      67 2777.35
   103.4 2765.78   123.6 2763.81   135.7  2760.9   144.6 2759.74   151.9 2759.56
     164 2760.85   188.2 2761.89   208.5 2761.11   214.7 2759.73   220.6 2758.41
   224.1  2758.4   232.7 2758.59   237.8 2759.57   244.8  2759.7   252.9 2759.08
     261 2760.71   281.4 2761.78   301.4  2762.2   305.5 2761.92   333.8 2762.87
   337.9 2764.09   341.9 2766.29   362.1  2779.6   374.2 2788.69   392.9 2799.98
#Mann= 5 ,-1,0
       0      .1       0     180     .08       0   214.7    .045       0
   237.8     .08       0     280      .1       0
Bank Sta=214.7,237.8
XS Rating Curve= 0 ,0
Exp/Cntr(USF)=0,0
Exp/Cntr=0.3,0.1

Type RM Length L Ch R = 1 ,11255   ,182.2,181,181
XS GIS Cut Line= 2
2306703.39612684551943.0183084032306701.38861857552292.324746539
#Sta/Elev= 30
       0 2796.22    10.2  2790.1    14.2 2787.39    34.2 2771.39    42.2 2764.07
    46.2 2762.27    54.2 2761.15    66.2  2760.8    90.2 2762.89   110.2 2761.81
   120.7 2762.69   126.2 2762.81   138.2 2761.91   156.92758.585   166.2 2757.14
   174.2 2757.16   183.62758.197   218.2 2760.86   246.2 2761.13   254.2 2760.22
   258.2  2760.9   262.2  2762.5   266.2 2763.12   274.2 2763.56   278.2 2764.11
   282.2 2766.09   291.7 2773.55   302.2 2779.93   319.6 2786.64   349.3 2798.87
#Mann= 5 ,-1,0
       0     .06       0     140     .08       0   156.9    .045       0
   183.6     .08       0     240     .06       0
Bank Sta=156.9,183.6
XS Rating Curve= 0 ,0
Exp/Cntr(USF)=0,0
Exp/Cntr=0.3,0.1

Type RM Length L Ch R = 1 ,11074   ,264.7,261.3,246.7
XS GIS Cut Line= 2
 2306526.7353995551934.9882753422306534.76543256552274.257172153
#Sta/Elev= 30
       0  2811.4    15.3  2803.8    30.2 2795.47    50.2 2783.27    62.2 2776.58
    70.2 2771.06    78.2    2765    82.2 2762.81    86.2 2761.64   102.2 2759.78
   114.2 2759.49   122.2 2759.34   130.2 2759.89   146.2 2760.31   186.2 2759.62
   194.2 2760.05   202.2 2759.63   214.3 2759.67   222.4 2758.48   230.2 2756.63
   234.2 2756.53   238.5 2756.98   246.3 2758.47   261.5 2761.81   275.3 2766.91
   286.3 2769.43   292.8 2771.53   310.3 2778.06   330.3 2786.66   339.4 2791.09
#Mann= 3 ,-1,0
       0      .1       0   222.4    .045       0   246.3      .1       0
Bank Sta=222.4,246.3
XS Rating Curve= 0 ,0
Exp/Cntr(USF)=0,0
Exp/Cntr=0.3,0.1

Type RM Length L Ch R = 1 ,10812   ,172.9,171.2,167.3
XS GIS Cut Line= 2
2306270.61778324551973.0337827522306367.15714203552271.909057899
#Sta/Elev= 30
       0 2801.99      17 2793.15    25.4 2790.28    33.8 2785.14    42.2 2781.06
    63.2 2773.04    67.4 2770.78      84 2760.24    87.1  2757.9      892756.944
    96.7 2755.58   109.2 2755.22   113.6 2755.33   117.9 2755.95     122  2757.2
   128.4 2758.56   134.7 2758.97   147.5 2757.91   153.9 2758.27   164.1  2759.7
   176.7 2760.14   189.3 2759.58   207.9 2759.96   235.5 2762.89   239.8 2763.61
     246 2765.29     286 2771.49   294.4 2773.75   303.2  2776.9   314.1 2781.46
#Mann= 3 ,-1,0
       0      .1       0      89    .045       0     122      .1       0
Bank Sta=89,122
XS Rating Curve= 0 ,0
Exp/Cntr(USF)=0,0
Exp/Cntr=0.3,0.1

Type RM Length L Ch R = 1 ,10641   ,193.8,200.6,210.9
XS GIS Cut Line= 3
2306078.86152264551958.4867560862306085.47380749552008.740120934
2306252.10338567 552353.90139002
#Sta/Elev= 30
       0 2805.98    18.9  2793.7    43.1 2773.58    51.2 2766.21      59 2761.81
    64.5 2759.53    68.9  2759.1    73.4 2760.34    77.8 2758.69   113.4 2758.36
   130.9 2759.09   153.3 2757.08   166.7 2758.59   176.5  2756.3   190.52755.856
   197.8 2753.74   211.1  2753.6   226.2 2755.33   273.3 2756.08   277.7 2756.38
   286.6 2758.65   295.5 2759.52   313.2 2758.32     331 2758.92   361.6 2758.33
   379.9 2758.99   384.3 2760.66   402.1 2772.47   419.8  2782.5     434 2787.54
#Mann= 6 ,-1,0
       0      .1       0  130.69     .08       0   190.5    .045       0
   226.2      .1       0  240.69     .08       0  350.69      .1       0
#XS Ineff= 2 , 0
                          296.14         2778.54
Permanent Ineff=
       F       F
Bank Sta=190.5,226.2
XS Rating Curve= 0 ,0
Exp/Cntr(USF)=0,0
Exp/Cntr=0.3,0.1

Type RM Length L Ch R = 1 ,10441   ,174.4,185.3,194.6
XS GIS Cut Line= 2
2305953.22811052552008.7401209342305966.45268021552341.999277293
#Sta/Elev= 30
       0 2789.67    20.5 2778.79    40.5 2771.21    48.5 2767.81    52.5 2765.37
    60.5  2759.4    64.5 2757.71    68.7  2757.2    89.1 2757.47   100.5 2757.01
   108.5 2757.38   132.5 2756.08   152.6 2756.53   156.6 2756.27   160.6 2755.33
   164.6  2754.1   176.5 2753.59   184.6 2753.87   193.3 2754.85   204.6 2755.34
   220.6 2758.38   244.6 2761.48   248.6 2762.44   252.6 2764.69   256.6 2765.98
   284.7 2767.02   289.2 2767.58   296.7 2769.17   315.1 2775.11   333.5 2780.21
#Mann= 3 ,-1,0
       0      .1       0   160.6    .045       0   193.3     .08       0
Bank Sta=160.6,193.3
XS Rating Curve= 0 ,0
Exp/Cntr(USF)=0,0
Exp/Cntr=0.3,0.1

Type RM Length L Ch R = 1 ,10255   ,230.3,216.2,200.8
XS GIS Cut Line= 2
2305869.59005417552007.5678689532305694.62899708552330.115123857
#Sta/Elev= 30
       0 2791.16      20 2782.84    33.7 2778.79    56.4 2769.72    61.2 2768.31
    79.2 2765.65    92.8 2764.88   106.5 2764.78   111.4 2763.48   120.2  2758.3
   126.1 2756.28   137.9 2755.24     152 2755.42   161.1 2754.61   165.7 2755.04
   170.8 2754.84   179.1 2753.04   182.2 2753.02     191 2753.44   197.5 2755.15
   211.2 2758.33   215.7 2758.96   247.6  2761.7   274.9 2761.62   279.6 2761.88
   297.6 2764.66   315.8 2764.78   341.5 2771.91   356.8 2774.55   366.9 2775.56
#Mann= 4 ,-1,0
       0      .1       0   170.8    .045       0   197.5      .1       0
     200     .08       0
Bank Sta=170.8,197.5
XS Rating Curve= 0 ,0
Exp/Cntr(USF)=0,0
Exp/Cntr=0.3,0.1

Type RM Length L Ch R = 1 ,10039   ,310.2,317.7,327.2
XS GIS Cut Line= 3
 2305557.1237672551941.6227993212305545.22165447552038.162158107
2305645.72838417552318.523035679
#Sta/Elev= 30
       0 2779.68     7.6 2778.97    18.4 2776.71    27.8 2775.38    47.9 2770.52
    68.1 2770.01    79.4  2769.1    92.2 2767.15   113.2 2764.75     126 2761.37
   130.2 2760.83   153.4 2761.79   181.2 2760.47   202.5  2757.5   212.7 2753.37
   215.2 2752.41   219.5 2751.64     228 2751.67   236.4 2753.25   253.4 2753.45
   270.8 2754.48   283.2 2755.72   321.4 2755.02   334.2 2757.38   346.9  2758.1
   351.2 2759.89   363.9  2767.2   380.9 2775.13   386.6  2776.9   395.1 2778.49
#Mann= 4 ,-1,0
       0      .1       0   212.7    .045       0   236.4      .1       0
  247.27     .08       0
Bank Sta=212.7,236.4
XS Rating Curve= 0 ,0
Exp/Cntr(USF)=0,0
Exp/Cntr=0.3,0.1

Type RM Length L Ch R = 1 ,9721    ,272.6,260,252.8
XS GIS Cut Line= 4
2305387.84927508551962.7821108362305401.07384478552024.937588411
2305353.46539387552367.453943557 2305382.5594472552412.417480526
#Sta/Elev= 30
       0 2776.54      27 2775.81    47.4 2773.21    64.6 2772.76    71.9 2771.61
    75.9 2769.01    89.4 2757.79  101.44 2751.09   108.2 2750.14   124.4 2751.08
   144.6 2752.47   156.7 2754.72   205.1 2755.59   253.6 2753.42   277.8 2754.08
   289.9 2753.05   306.1 2753.96   339.5 2753.81   346.5 2753.24   354.6  2750.5
   358.8 2750.74   374.8 2752.46   386.9 2757.34   390.9 2757.28   394.9 2755.62
     399 2755.38   407.1 2756.74   415.5 2761.03   435.7 2773.81   462.9 2777.62
#Mann= 6 ,-1,0
       0      .1       0  101.44    .045       0   124.4      .1       0
  343.55     .08       0  419.36      .1       0  429.36     .08       0
Bank Sta=101.44,124.4
XS Rating Curve= 0 ,0
Exp/Cntr(USF)=0,0
Exp/Cntr=0.3,0.1

Type RM Length L Ch R = 1 ,9461    ,263.7,272.9,273.4
XS GIS Cut Line= 3
2305088.97399994551961.4596538662305100.87611266552034.194787198
2305271.47306175552430.931878102
#Sta/Elev= 30
       0 2786.97      20 2777.23    32.1 2774.27    44.3 2769.14    60.5 2764.32
      77 2756.56    98.7 2750.08     151 2750.74   157.1  2749.9     164 2748.34
   168.4 2748.17   177.1 2748.21   190.2 2749.58   213.7 2750.56   238.1 2748.36
   256.4 2749.49   312.1  2749.8   329.5 2751.31   346.9 2751.65   355.6 2750.81
   364.3 2751.96   377.4 2750.78   403.5 2749.98   442.7 2751.78     456 2754.01
   464.5 2754.35   473.2 2756.06   477.4 2757.54   486.2  2763.6   505.6 2773.19
#Mann= 5 ,-1,0
       0      .1       0   157.1    .045       0   190.2      .1       0
   243.7     .08       0   453.7      .1       0
Bank Sta=157.1,190.2
XS Rating Curve= 0 ,0
Exp/Cntr(USF)=0,0
Exp/Cntr=0.3,0.1

Type RM Length L Ch R = 1 ,9188    ,328.7,350.6,364
XS GIS Cut Line= 2
2304866.44204319552014.080379956 2304988.8917626552459.797358625
#Sta/Elev= 30
       0 2780.73    15.7 2773.19    28.1 2766.39    36.4 2763.53    48.8 2760.64
    72.3 2757.74    88.5 2753.18   102.8 2750.78   119.4 2750.77   148.4 2752.45
   156.9 2751.03   169.1 2747.83   173.3 2746.91   185.7 2746.83   192.7 2748.08
   198.2 2748.77   210.6    2748   270.8 2749.55   293.6 2748.03   322.6 2749.11
   339.2 2747.75     360 2749.92   385.2 2750.73   401.4 2754.18   409.7 2754.15
   413.9 2755.37   426.3  2762.5   434.6 2765.07   451.2 2772.25   462.2 2775.83
#Mann= 4 ,-1,0
       0      .1       0   169.1    .045       0   192.7     .08       0
     280      .1       0
Bank Sta=169.1,192.7
XS Rating Curve= 0 ,0
Exp/Cntr(USF)=0,0
Exp/Cntr=0.3,0.1

Type RM Length L Ch R = 1 ,8838    ,267.5,264.5,262.8
XS GIS Cut Line= 4
2304796.07681478552026.139600897  2304794.286011552077.806089042
2304594.61348992552338.5189523122304588.98005333552375.154476531
#Sta/Elev= 30
       0 2776.86      11 2771.05    39.1 2758.71    51.7 2755.35    55.9 2753.73
      66 2748.21    71.1 2746.93    76.1 2746.45    86.2  2747.3     107 2747.11
   136.6 2748.02   181.9 2746.31   213.1 2748.12   217.2 2747.66   222.2 2744.99
   226.8  2744.1   239.4 2745.39   259.1 2744.26   267.6 2745.44   277.6 2747.54
   297.8 2747.86   307.9 2750.81   311.7 2751.11   333.1 2751.38   353.2 2750.61
   368.3 2752.09   375.2 2754.51   390.9 2761.52   411.1 2773.19   417.2 2776.04
#Mann= 7 ,-1,0
       0      .1       0    61.7     .08       0    91.7      .1       0
   181.7     .08       0   239.4    .045       0   267.6     .08       0
   311.7      .1       0
#XS Ineff= 2 , 0
                          311.11         2759.32
Permanent Ineff=
       F       F
Bank Sta=239.4,267.6
XS Rating Curve= 0 ,0
Exp/Cntr(USF)=0,0
Exp/Cntr=0.3,0.1

Type RM Length L Ch R = 1 ,8573    ,247,250.5,259
XS GIS Cut Line= 2
2304568.31565282551949.4786760262304379.07206046552294.639945111
#Sta/Elev= 30
       0 2795.74    17.9 2786.75    54.4 2769.26    63.5 2763.49    77.2  2751.4
    85.3 2747.36    95.5 2743.74   113.7 2745.47   131.9 2744.96   138.4 2745.61
   154.8 2745.66     173 2746.95   182.1 2746.73   191.3 2745.45   195.8 2745.28
     215 2746.25   227.7 2744.69   241.3 2744.29   253.3 2743.08   265.1 2743.53
   270.9 2744.45   291.6 2747.44   300.7 2746.09   323.5 2748.75   350.5 2750.15
   355.5 2751.16   364.6 2754.23   373.7 2759.12     383 2762.55   393.6 2765.28
#Mann= 5 ,-1,0
       0      .1       0     190     .12       0   241.3    .045       0
   270.9     .08       0     380      .1       0
#XS Ineff= 2 , 0
                          294.11         2761.41
Permanent Ineff=
       F       F
Bank Sta=241.3,270.9
XS Rating Curve= 0 ,0
Exp/Cntr(USF)=0,0
Exp/Cntr=0.3,0.1

Type RM Length L Ch R = 1 ,8323    ,226.5,231,235.3
XS GIS Cut Line= 2
2304396.92522955551872.1149432992304251.71945428552163.716705113
#Sta/Elev= 30
       0 2799.16    10.7 2793.41    50.3 2766.77    63.7 2758.21    84.9  2747.8
   92.71 2743.35      95 2742.29    99.5 2741.89   105.8 2743.17   108.7 2744.13
   112.9 2744.84   126.3 2744.96   135.2 2745.44   141.6 2745.26   157.6  2746.2
   172.2 2746.12   175.5 2746.27   184.4 2747.65   193.3 2748.17   207.2 2748.18
   211.2 2748.74   220.1 2751.08   242.5 2752.14   251.9 2755.41   269.3 2758.69
   278.2 2760.03   287.7 2761.02   296.1 2761.44   300.6 2762.14   325.8  2763.6
#Mann= 4 ,-1,0
       0      .1       0      50     .12       0   92.71    .045       0
   105.8     .12       0
Bank Sta=92.71,105.8
XS Rating Curve= 0 ,0
Exp/Cntr(USF)=0,0
Exp/Cntr=0.3,0.1

Type RM Length L Ch R = 1 ,8092    ,211.6,218.8,223.7
XS GIS Cut Line= 2
 2304215.0017304551770.2403522782304031.82821553552023.791059704
#Sta/Elev= 30
       0 2786.15       7 2783.82     9.9 2782.59    18.4 2777.67    28.3 2773.55
      39  2767.3      50  2761.8    55.7 2757.73    67.8 2747.57      70 2745.94
    73.1  2744.1    77.6 2743.32    92.4 2741.57    97.4 2741.72   102.3 2742.55
   104.4 2742.56   114.1 2741.66   141.4 2740.75   146.7 2741.84   153.1 2744.45
   161.5 2746.34   187.5 2747.86   210.9 2747.71   240.5 2748.94   250.5 2750.55
   260.2 2751.47   270.1 2754.38     280  2756.2   304.9 2758.76   312.8 2759.32
#Mann= 5 ,-1,0
       0      .1       0   114.1    .045       0   146.7      .1       0
     230     .08       0     270      .1       0
Bank Sta=114.1,146.7
XS Rating Curve= 0 ,0
Exp/Cntr(USF)=0,0
Exp/Cntr=0.3,0.1

Type RM Length L Ch R = 1 ,7873    ,363,369.9,378
XS GIS Cut Line= 2
2304088.70841225551648.7673897862303819.73256673 551857.97082519
#Sta/Elev= 30
       0 2764.08      26 2750.96    31.1 2748.08    36.1 2745.88    41.2 2744.25
    60.5 2743.54    71.6 2743.89    80.5 2742.45    94.7 2740.88     102 2740.06
   114.7 2739.36   117.5 2739.44   127.4  2740.9   137.5 2742.03   170.1 2741.67
   183.1    2740   188.8 2739.69   197.4 2740.19   211.6 2741.82   223.6 2740.56
   233.8 2741.44   243.9  2741.8   254.4 2743.79   282.9 2750.31   294.6 2751.01
   299.7  2751.8   308.5 2756.24   314.2 2757.99   330.1 2761.75   340.8 2765.34
#Mann= 5 ,-1,0
       0      .1       0    94.7    .045       0   127.4      .1       0
     140     .08       0     230      .1       0
#XS Ineff= 2 , 0
           70.68 2751.91
Permanent Ineff=
       F       F
Bank Sta=94.7,127.4
XS Rating Curve= 0 ,0
Exp/Cntr(USF)=0,0
Exp/Cntr=0.3,0.1

Type RM Length L Ch R = 1 ,7503    ,235,238.8,244.1
XS GIS Cut Line= 2
2304056.60461779551408.5400099042303633.40261816551489.700830847
#Sta/Elev= 30
       0 2764.44    16.7    2758    45.2 2745.16    57.5  2741.6    73.7 2739.22
   118.6 2738.44   130.8 2739.62   155.2 2738.55   171.5 2739.45   204.1 2739.55
   224.4 2737.12   240.7 2738.35     257 2737.91   289.6 2738.67   314.1 2737.75
   322.42736.252   330.3 2735.12   338.5 2734.93   343.2 2735.09   347.92736.444
   350.7 2737.92   358.9 2740.29   362.9 2742.33     367 2746.28   371.1  2752.9
   375.1 2758.38   387.4 2770.01   411.8 2787.67     424 2793.68   430.9 2799.08
#Mann= 5 ,-1,0
       0      .1       0      80     .08       0   322.4    .045       0
   347.9     .08       0     380      .1       0
#XS Ineff= 2 , 0
          180.68 2750.15
Permanent Ineff=
       F       F
Bank Sta=322.4,347.9
XS Rating Curve= 0 ,0
Exp/Cntr(USF)=0,0
Exp/Cntr=0.3,0.1

Type RM Length L Ch R = 1 ,7264    ,176.7,169.4,164.7
XS GIS Cut Line= 4
2303993.14959143551189.1748583222303914.90879955551243.220731081
 2303689.9272049551230.9237749262303599.99485174 551272.24603045
#Sta/Elev= 30
       0 2764.47    10.9 2759.47    40.1 2747.53    49.8 2744.18    66.8 2739.59
    81.2 2738.61   113.9  2739.6   153.9 2738.22   161.9 2737.16   165.9 2735.68
   169.9 2734.87     182  2735.2     194 2736.24   213.6  2735.6     234 2736.87
   252.6 2734.56   258.1 2733.04   270.6 2734.01   282.1 2733.41   294.1 2733.73
   302.1 2735.43   331.1 2738.13   335.7 2741.03   353.2 2757.64   362.6 2763.82
   371.7 2768.49   384.5 2775.89   392.8 2779.49   401.6 2784.08   419.4 2790.27
#Mann= 5 ,-1,0
       0      .1       0  125.09     .08       0   252.6    .045       0
   270.6     .08       0  320.41      .1       0
Bank Sta=252.6,270.6
XS Rating Curve= 0 ,0
Exp/Cntr(USF)=0,0
Exp/Cntr=0.3,0.1

Type RM Length L Ch R = 1 ,7095    ,381.5,372.7,367.8
XS GIS Cut Line= 3
2303911.37681137550958.3826035652303871.60364029551019.411519721
2303589.22173108551113.502243631
#Sta/Elev= 30
       0 2772.46    24.6 2764.57    50.6 2755.52    55.9 2754.79    65.4 2754.58
      77 2752.91    97.5 2748.79   102.3 2746.63   114.4 2737.94   118.6 2736.28
   131.3 2735.17   156.6 2734.37   194.5 2731.99   198.7 2731.99   207.2 2733.05
   211.4 2733.02   217.6 2732.09   240.9 2731.08   247.92731.385   260.4 2732.16
   270.4  2734.9   274.6 2735.51   293.5 2735.47     311 2734.66   316.8 2735.73
     321 2737.59   333.1 2744.64   364.7 2764.84   367.4 2766.32   370.5 2766.77
#Mann= 3 ,-1,0
       0      .1       0   217.6    .045       0   247.9      .1       0
Bank Sta=217.6,247.9
XS Rating Curve= 0 ,0
Exp/Cntr(USF)=0,0
Exp/Cntr=0.3,0.1

Type RM Length L Ch R = 1 ,6722    ,322,308.3,301.3
XS GIS Cut Line= 2
2303690.98193839 550682.645762912303460.08095149550943.302031634
#Sta/Elev= 30
       0 2791.59    10.3 2786.52    16.3 2782.14    26.5 2773.14    34.4 2767.29
    51.5 2751.53    60.5 2742.53    64.6 2737.63    67.5 2733.42      69 2731.94
    70.6 2730.72    74.6 2729.17    80.3 2728.39    94.2 2728.96    99.6 2728.66
   108.6 2730.52   124.9 2729.67   131.6 2731.71   136.9 2732.25   148.3 2731.83
   156.8 2729.87   159.6 2729.71   174.4 2731.16     222 2731.97   239.5 2733.07
   270.6 2732.37   291.9 2732.86   318.7  2741.8   329.6 2747.08   348.2 2754.46
#Mann= 4 ,-1,0
       0      .1       0    74.6    .045       0    94.2      .1       0
     300     .08       0
#XS Ineff= 2 , 0
                          242.58         2743.72
Permanent Ineff=
       F       F
Bank Sta=74.6,94.2
XS Rating Curve= 0 ,0
Exp/Cntr(USF)=0,0
Exp/Cntr=0.3,0.1

Type RM Length L Ch R = 1 ,6414    ,286.2,286.5,285.5
XS GIS Cut Line= 2
2303332.72834531550599.3309738212303327.96750022550890.932735635
#Sta/Elev= 30
       0 2777.41    13.5 2769.02    21.9 2764.45    41.9 2752.49    45.9 2750.39
    53.9 2747.12    65.9 2740.37    81.9 2730.58    93.9 2726.44   104.7 2725.66
   109.9 2724.98   125.9  2724.8   133.42724.874   137.9 2724.86   145.9 2725.95
   153.9 2726.06   165.9 2727.55   173.9 2727.74   185.9 2728.59   193.9 2730.65
   197.9 2731.24   213.9  2731.6   226.7 2730.48   233.9 2730.36   241.9 2731.49
   249.4 2731.32   253.9 2731.62   257.9 2732.56   261.9 2734.53   291.6 2752.14
#Mann= 4 ,-1,0
       0      .1       0   104.7    .045       0   133.4      .1       0
     210     .08       0
#XS Ineff= 2 , 0
                          210.33         2744.27
Permanent Ineff=
       F       F
Bank Sta=104.7,133.4
XS Rating Curve= 0 ,0
Exp/Cntr(USF)=0,0
Exp/Cntr=0.3,0.1

Type RM Length L Ch R = 1 ,6127    ,271.9,273.2,274
XS GIS Cut Line= 2
2303057.78954131550589.8092836392303056.59933004550824.280904363
#Sta/Elev= 30
       0 2764.79     7.4 2760.62    15.4 2757.51    27.4 2751.71    31.4 2750.11
    43.4 2743.95      54    2739    67.4 2733.63    71.4 2732.64    79.4 2729.71
    83.4 2728.52    87.4 2727.86   103.4 2726.52   111.4 2725.22   119.4 2724.33
   124.4 2723.18   127.4 2722.38   131.4  2721.9   135.4 2722.17   143.4 2721.62
   156.2 2722.58   171.4 2723.59   175.4  2724.5   180.1 2727.02   187.4 2731.63
     200 2741.12   207.4  2745.3   219.4  2752.6   227.8 2757.04   234.5 2760.26
#Mann= 5 ,-1,0
       0      .1       0     120     .08       0   124.4    .045       0
   156.2     .08       0     220      .1       0
Bank Sta=124.4,156.2
XS Rating Curve= 0 ,0
Exp/Cntr(USF)=0,0
Exp/Cntr=0.3,0.1

Type RM Length L Ch R = 1 ,5854    ,302.3,301.9,302
XS GIS Cut Line= 2
2302794.50539663  550529.50537712302781.02339663 550786.99527206
#Sta/Elev= 30
       0 2768.66     7.7 2765.44    19.7 2761.01    36.2 2753.75      40 2751.96
    59.8 2741.14    71.8 2735.67    79.8 2731.56    89.4 2728.24    97.1 2725.99
   111.8 2720.11   115.8 2719.69   119.9  2720.3   123.8 2721.42   127.8 2722.13
   135.9 2722.78   143.9  2721.6   151.9 2721.27   167.9 2718.04   169.72717.939
   179.9 2717.33   200.1 2718.12     204 2719.63     208 2722.24     220 2731.47
     228 2736.05     236 2738.84     248 2744.23     252 2745.62   257.8 2745.94
#Mann= 3 ,-1,0
       0      .1       0   169.7    .045       0   200.1      .1       0
Bank Sta=169.7,200.1
XS Rating Curve= 0 ,0
Exp/Cntr=0.3,0.1

Type RM Length L Ch R = 1 ,5552    ,254.7,262.3,266.4
XS GIS Cut Line= 2
2302489.46449409 550533.539341472302482.32322646 550793.00539892
#Sta/Elev= 30
       0 2754.31    10.6 2751.34    14.8 2749.79    23.6 2745.27    39.7 2738.86
    59.7 2729.73    67.7 2726.81    91.7  2720.7    99.7 2717.54   103.7 2716.51
   111.7 2716.52   115.7 2716.05   119.7  2714.8   123.7 2714.01   127.7 2713.86
   131.32713.885   147.7 2714.14   155.7 2714.59   171.7 2715.79   183.7 2718.47
   199.5 2719.95   203.7 2720.69   211.7 2723.09   223.7  2728.2   227.7 2729.65
   235.7 2730.75   239.7 2732.02   243.7 2734.41   247.7 2736.12   259.6 2740.11
#Mann= 3 ,-1,0
       0      .1       0   131.3    .045       0   155.7      .1       0
Bank Sta=131.3,155.7
XS Rating Curve= 0 ,0
Exp/Cntr(USF)=0,0
Exp/Cntr=0.3,0.1

Type RM Length L Ch R = 1 ,5290    ,277.6,287.3,297.3
XS GIS Cut Line= 2
2302293.25514037550454.7970432692302169.24766146550808.122197816
#Sta/Elev= 30
       0 2738.47    24.7 2733.27    49.2 2727.41    57.6 2726.29    78.8 2713.95
    83.1 2712.24    95.8 2711.93   100.1 2712.54   155.1 2715.43   159.4  2714.4
   163.6  2711.9   167.9 2710.31     1712710.001   184.8 2709.78   201.8 2710.41
     213 2712.23     223 2711.59   248.4 2713.43   261.1 2712.87   269.6 2711.44
   282.3 2712.39   291.4 2712.47     295 2713.85   297.7 2715.75   307.7 2724.39
   328.9 2739.07   358.6 2756.65   362.9 2759.48   369.8 2764.99   374.5 2767.28
#Mann= 3 ,-1,0
       0      .1       0     171    .045       0   201.8      .1       0
#XS Ineff= 2 , 0
          149.57 2732.15
Permanent Ineff=
       F       F
Bank Sta=171,201.8
XS Rating Curve= 0 ,0
Exp/Cntr=0.3,0.1

Type RM Length L Ch R = 1 ,5003    ,305.6,307.8,310.7
XS GIS Cut Line= 2
2302144.43902964 550376.906940682301900.51918856550591.438849094
#Sta/Elev= 30
       0  2730.1     8.9 2728.87    16.3 2726.46    23.1 2722.36    32.3 2715.02
    37.2 2711.83    42.8 2709.87    45.7 2709.49    54.9  2708.8    96.2  2709.9
   113.7 2710.82   122.9 2709.81   142.1 2710.27   163.9 2708.83   176.1 2709.78
   190.3 2709.44   201.6 2710.02   206.3 2709.87   212.4 2708.84   218.6 2707.05
   230.4 2705.65   254.8 2704.77  259.32 2705.64     264 2707.68   266.8 2709.82
     279 2722.32   303.6 2744.13   309.3 2747.75   314.6 2751.78   324.8 2757.65
#Mann= 5 ,-1,0
       0      .1       0     180     .08       0     200      .1       0
   230.4    .045       0  259.32      .1       0
#XS Ineff= 2 , 0
          176.23 2724.12
Permanent Ineff=
       F       F
Bank Sta=230.4,259.32
XS Rating Curve= 0 ,0
Exp/Cntr(USF)=0,0
Exp/Cntr=0.3,0.1

Type RM Length L Ch R = 1 ,4695    ,164.4,162.6,161.1
XS GIS Cut Line= 2
2301987.21358991550152.0892558352301710.96702291550343.110818122
#Sta/Elev= 30
       0 2721.25    28.8 2707.75    34.6 2706.11      49 2705.95    57.2 2705.47
    65.2 2704.25    81.5  2702.5     101 2704.26   109.3 2703.78   115.5 2704.41
   125.3 2703.23   139.9    2703   152.5 2703.08   164.2 2703.75     169 2703.58
   172.6 2702.89   178.3 2700.91   182.12700.703   192.7 2700.25   207.9 2700.98
     210 2701.24     234 2705.81   251.7 2707.15   276.1  2708.2   290.5 2711.55
   304.9 2719.51   313.5 2724.67   319.8 2727.26   324.7 2728.71   335.9 2734.29
#Mann= 5 ,-1,0
       0      .1       0      90     .08       0   182.1    .045       0
   207.9     .08       0     210      .1       0
#XS Ineff= 2 , 0
          102.55 2708.76
Permanent Ineff=
       F       F
Bank Sta=182.1,207.9
XS Rating Curve= 0 ,0
Exp/Cntr(USF)=0,0
Exp/Cntr=0.3,0.1

Type RM Length L Ch R = 1 ,4532    ,157.3,155.8,154.1
XS GIS Cut Line= 2
2301879.26908394550011.5994237252301626.97820175550220.224576309
#Sta/Elev= 30
       0 2718.19       4 2716.41    11.8 2713.95    19.6 2710.73    34.6 2706.25
    45.5 2702.19    48.8 2701.65    61.1 2701.94    66.3 2701.39    71.5 2700.09
    81.9 2700.15    90.4 2698.73   123.4 2698.37   149.3 2700.37   159.6 2700.31
   170.1 2699.09   176.6  2698.1   185.1 2697.82   197.82698.875   210.7 2698.87
   230.6 2701.22   244.8 2701.08     248 2701.22   258.3 2702.77   276.1 2702.88
   284.3 2703.51   289.5  2705.8   301.6 2713.06   315.4 2718.82   327.4 2726.23
#Mann= 3 ,-1,0
       0      .1       0   170.1    .045       0   197.8      .1       0
Bank Sta=170.1,197.8
XS Rating Curve= 0 ,0
Exp/Cntr(USF)=0,0
Exp/Cntr=0.3,0.1

Type RM Length L Ch R = 1 ,4376    ,259.9,255.3,251.2
XS GIS Cut Line= 2
2301766.80409496549887.5978619012301522.88425389550121.231926543
#Sta/Elev= 30
       0 2726.63     9.2 2723.54    25.6 2716.09    39.8 2711.18    53.9 2705.57
    65.2 2700.42      68 2699.63    77.5 2699.08   112.2  2698.8   127.5 2696.05
   135.3  2695.3   142.1  2695.7   152.6 2697.26   158.6 2697.01   169.8 2695.35
   175.3 2695.12   186.9 2695.51   195.4 2697.03     203 2698.64   208.6 2699.01
     218 2698.99   241.8 2697.74   254.8 2698.36   277.4 2697.68   283.1 2698.48
   302.9 2706.52   308.3 2710.57   320.3 2721.71   331.9 2730.23   337.8 2733.86
#Mann= 4 ,-1,0
       0      .1       0   158.6    .045       0   195.4     .08       0
     200      .1       0
Bank Sta=158.6,195.4
XS Rating Curve= 0 ,0
Exp/Cntr(USF)=0,0
Exp/Cntr=0.3,0.1

Type RM Length L Ch R = 1 ,4121    ,309.7,308.6,290
XS GIS Cut Line= 2
2301552.27218655549693.6375063492301355.37303773549968.414676714
#Sta/Elev= 30
       0 2720.03    14.2 2715.28    19.1 2714.14    34.1 2707.83    42.7 2704.87
    73.3 2698.88    83.1 2694.02      88 2693.73   102.9 2694.59   112.6 2694.29
   127.4 2692.61   142.1 2693.91   166.7  2693.6   171.8 2693.08   176.6 2691.73
   178.7 2691.62   196.3 2691.95     209 2693.29   219.9 2694.44   231.9 2694.04
   243.4 2694.59   254.3 2693.67   265.2 2691.99   272.1 2692.57   277.8 2694.02
   279.9 2694.94   281.7 2696.34   304.5 2717.94   334.1 2740.92     338  2743.5
#Mann= 5 ,-1,0
       0      .1       0     160     .08       0   171.8    .045       0
     209     .08       0     280      .1       0
Bank Sta=171.8,209
XS Rating Curve= 0 ,0
Exp/Cntr(USF)=0,0
Exp/Cntr=0.3,0.1

Type RM Length L Ch R = 1 ,3813    ,230.9,228,226
XS GIS Cut Line= 2
2301270.14803302549523.187496924 2301193.7394081 549902.29182823
#Sta/Elev= 30
       0 2716.96       2 2715.49    10.2 2713.44    14.3 2711.58    26.5  2703.4
    46.9 2694.17    59.2 2690.44    75.5 2688.44    91.8 2689.54   112.2 2688.42
   124.4 2688.86   144.8 2687.02   148.9  2687.2   161.2  2689.9   177.5  2689.1
   185.7 2690.62   193.8 2691.09   206.1 2688.92   222.4 2688.77   230.5 2690.27
   246.9 2689.28   258.1 2690.02   267.3 2688.07   283.6 2686.47   295.8 2686.65
   298.8 2688.21   320.3 2705.75   332.5 2714.36   356.5 2726.63   386.7 2740.16
#Mann= 3 ,-1,0
       0      .1       0   267.3    .045       0   298.8      .1       0
#XS Ineff= 2 , 0
          127.58 2699.87
Permanent Ineff=
       F       F
Bank Sta=267.3,298.8
XS Rating Curve= 0 ,0
Exp/Cntr(USF)=0,0
Exp/Cntr=0.3,0.1

Type RM Length L Ch R = 1 ,3585    ,191,183.5,174
XS GIS Cut Line= 4
2301099.69802359549467.3504248712301001.24844918549571.677585812
2300983.51362442549841.7661856492301005.65663908549889.067258534
#Sta/Elev= 30
       0 2728.29       8 2726.26      52 2709.98    57.6 2708.92      74 2702.93
    86.7 2699.63   114.1 2693.93   127.5 2693.62   139.2 2694.83   144.9 2694.44
     149 2693.93   168.4 2689.09     177 2688.45     189 2688.66   201.1 2686.79
   220.9 2688.81   259.7 2686.45   281.3 2687.34   292.6 2687.02   297.3 2686.66
   305.3 2682.36   309.3  2681.4   325.3 2682.03   333.4 2681.15   341.4 2680.72
   353.52680.842   361.4 2681.27   385.5 2685.74   420.2  2703.8   466.3 2723.69
#Mann= 3 ,-1,0
       0      .1       0   333.4    .045       0   353.5      .1       0
Bank Sta=333.4,353.5
XS Rating Curve= 0 ,0
Exp/Cntr(USF)=0,0
Exp/Cntr=0.3,0.1

Type RM Length L Ch R = 1 ,3401    ,239.6,241.3,243.1
XS GIS Cut Line= 2
2300684.86329394549565.2656488622300885.68083378549937.512795882
#Sta/Elev= 30
       0 2693.28    20.1 2693.46    49.9 2692.29    61.4 2690.88    68.1 2688.99
    82.1 2686.72    93.9 2687.06   108.1 2686.52   118.1 2687.29   127.2 2686.07
   145.3 2687.33   168.1 2685.68   181.7 2682.62   234.4 2683.24   240.8 2682.58
   254.4  2679.7   268.1  2678.1   268.1 2678.09   277.1 2677.06   288.72678.103
   297.6 2678.99     309 2681.22   321.2  2682.1   349.9 2688.62   363.5 2697.67
   372.6 2702.24   377.1 2705.92   386.2 2711.94   408.9 2723.84     423 2730.21
#Mann= 4 ,-1,0
       0     .06       0      70      .1       0   268.1    .045       0
   288.7      .1       0
#XS Ineff= 2 , 0
           231.3 2691.81
Permanent Ineff=
       F       F
Bank Sta=268.1,288.7
XS Rating Curve= 0 ,0
Exp/Cntr(USF)=0,0
Exp/Cntr=0.3,0.1

Type RM Length L Ch R = 1 ,3160    ,265.1,265.5,267
XS GIS Cut Line= 2
2300503.12299061 549674.535350122300645.65446401550028.659938666
#Sta/Elev= 30
       0  2686.2      33 2683.62    41.7 2682.44    50.3 2680.44    58.9 2679.49
    71.8 2679.18    89.1  2680.4   106.3 2679.56     115 2677.94   119.7 2678.98
   132.2 2678.05   140.8 2678.69   162.4 2677.75   179.6 2678.05   188.3 2679.32
   196.9 2678.53   218.4 2678.44   231.4  2676.7   242.6  2673.8   248.12673.267
   261.6 2672.85   271.42673.706   274.5 2674.16   283.1  2676.8   296.1 2678.21
   300.4 2680.27   334.8  2704.9   347.2 2712.76     365 2724.94   381.7 2734.81
#Mann= 3 ,-1,0
       0      .1       0   248.1    .045       0   271.4      .1       0
#XS Ineff= 2 , 0
          189.29 2686.33
Permanent Ineff=
       F       F
Bank Sta=248.1,271.4
XS Rating Curve= 0 ,0
Exp/Cntr(USF)=0,0
Exp/Cntr=0.3,0.1

Type RM Length L Ch R = 1 ,2894    ,274.8,272.2,272.5
XS GIS Cut Line= 2
2300235.92001211549676.6963773742300407.67349702550165.190055228
#Sta/Elev= 30
       0 2687.38    13.1 2684.72    51.4 2680.22    59.9 2680.36    72.6 2678.77
    88.4 2679.95   102.3 2679.33   110.8 2677.87   119.2  2675.1   123.5 2674.65
     132  2675.1   145.5 2677.11   216.8 2676.96   225.2 2675.94   233.7 2674.03
   293.1 2673.24   301.6 2672.06   305.8 2672.29   314.3 2670.72   336.2 2672.19
     360 2670.63   377.9 2670.19   386.7 2670.34   390.6 2671.11   399.1 2675.72
   411.8 2678.83   420.3 2681.97   462.7 2703.95   500.8 2727.89   517.8 2737.11
#Mann= 4 ,-1,0
       0     .06       0      50      .1       0     360    .045       0
   386.7      .1       0
Bank Sta=360,386.7
XS Rating Curve= 0 ,0
Exp/Cntr(USF)=0,0
Exp/Cntr=0.3,0.1

Type RM Length L Ch R = 1 ,2622    ,200.4,201.5,201.9
XS GIS Cut Line= 2
2299997.24958504549723.5382368952300157.85024625 550207.57078527
#Sta/Elev= 30
       0  2699.2    14.4 2692.59    22.8 2690.47    32.1 2684.94    52.3 2677.81
    69.2    2675    73.4 2673.41      86 2670.49   107.1 2667.71   115.5 2667.71
   123.9 2670.94   170.3 2667.13     184 2668.73   199.8 2668.59   212.5 2669.41
   263.1 2669.68   280.62668.377   296.7 2666.64   313.9 2668.01   347.3 2668.39
     360 2669.73   397.9 2670.19   406.3 2669.56     419 2670.54   427.4 2672.15
   443.5 2682.78     453 2690.04     478 2705.41   494.8 2716.41     510 2727.51
#Mann= 6 ,-1,0
       0     .06       0     100     .12       0     170      .1       0
     210     .12       0   280.6    .045       0   313.9      .1       0
Bank Sta=280.6,313.9
XS Rating Curve= 0 ,0
Exp/Cntr(USF)=0,0
Exp/Cntr=0.3,0.1

Type RM Length L Ch R = 1 ,2421    ,297.2,310.2,319.2
XS GIS Cut Line= 2
2299822.79234954549811.1892369862299941.81347681550207.926327889
#Sta/Elev= 30
       0 2691.06     6.3 2686.21      22 2676.63    43.8  2665.6    50.9  2664.3
    64.7 2664.12    95.9 2664.91   114.3 2666.11   127.4 2665.63   152.4 2666.33
   185.8 2666.38   198.4 2667.15   223.4 2665.45   240.4 2665.76   246.9 2665.34
     261 2664.31   273.5 2664.24   281.9 2665.45   298.2    2667   306.9 2666.35
   319.5 2667.09   327.8 2665.88     332 2665.92   340.3 2667.14     357 2668.18
   373.8  2671.4   381.8 2674.76   390.5  2679.8   394.6 2682.44   414.2 2697.22
#Mann= 6 ,-1,0
       0     .06       0      10      .1       0     100     .12       0
     110      .1       0   246.9    .045       0   281.9      .1       0
Bank Sta=246.9,281.9
XS Rating Curve= 0 ,0
Exp/Cntr(USF)=0,0
Exp/Cntr=0.3,0.1

Type RM Length L Ch R = 1 ,2110    ,292.7,291.3,276.3
XS GIS Cut Line= 3
2299654.55101504549862.5188360982299577.18728232550142.218485184
2299602.18171904550233.864753182
#Sta/Elev= 30
       0 2689.04    19.4 2676.42    31.8 2666.97      36 2664.49    49.6 2661.01
    56.7 2659.62    60.9  2659.4      65 2659.45    73.3 2660.74    95.1 2659.89
   115.1 2661.45   124.4 2661.31     159 2662.83   176.4 2662.28   185.4 2663.04
   193.7 2661.34   199.2 2660.84   218.6 2660.34   222.7 2661.48   226.9 2662.91
     231 2663.34   260.1  2662.8   280.4 2663.25   297.4 2662.03   311.3 2662.52
   327.6 2664.93   335.8  2667.2   351.3 2672.06   367.9 2678.61   385.2 2684.48
#Mann= 6 ,-1,0
       0     .06       0      60      .1       0   199.2    .045       0
   222.7      .1       0     260     .05       0   370.2      .1       0
Bank Sta=199.2,222.7
XS Rating Curve= 0 ,0
Exp/Cntr(USF)=0,0
Exp/Cntr=0.3,0.1

Type RM Length L Ch R = 1 ,1819    ,258.1,258,257.3
XS GIS Cut Line= 2
2299334.38418268549937.5021462782299437.93256341550267.190668818
#Sta/Elev= 30
       0 2692.63     3.9  2690.5    12.2 2684.86    20.6 2676.73      29  2669.5
    33.2 2666.58      49 2660.26    59.4 2656.99    62.6    2656    66.7 2655.44
    70.9 2655.48    77.7 2656.62   112.8 2660.15   133.8 2658.51   157.5 2659.55
   184.1 2658.91   213.5 2660.79   226.1 2661.03   238.6 2661.11   251.2 2660.12
   259.6 2660.12     268  2659.3   276.4 2659.34     289 2660.72   293.1  2661.6
   299.7  2664.5   313.8 2673.93   326.8 2680.66   335.1 2683.71   345.6 2686.43
#Mann= 3 ,-1,0
       0      .1       0    59.4    .045       0    77.7      .1       0
Bank Sta=59.4,77.7
XS Rating Curve= 0 ,0
Exp/Cntr(USF)=0,0
Exp/Cntr=0.3,0.1

Type RM Length L Ch R = 1 ,1561    ,239.4,238.8,238.3
XS GIS Cut Line= 2
 2299093.9615056550036.2896819132299190.36861869550315.989330999
#Sta/Elev= 30
       0 2681.95     5.6 2678.59     9.4  2675.8    19.1 2666.18    26.3 2657.95
    30.6 2653.89    34.8  2652.8    38.82652.468    52.8 2652.09    59.1 2652.13
    68.32652.768    77.1 2653.89    85.6  2655.7    89.8 2656.21      94 2656.34
    98.3 2655.51   102.5 2655.25   132.1 2654.73   144.8 2654.84   157.5  2655.8
   174.4 2656.49   182.9 2657.93   195.6  2659.2   215.5 2663.92   225.8 2666.05
   233.6 2668.21   254.8 2672.81   266.7 2677.25   271.7 2678.71   295.8 2688.26
#Mann= 3 ,-1,0
       0      .1       0    38.8    .045       0    68.3      .1       0
Bank Sta=38.8,68.3
XS Rating Curve= 0 ,0
Exp/Cntr(USF)=0,0
Exp/Cntr=0.3,0.1

Type RM Length L Ch R = 1 ,1322    ,236.5,235.7,234.8
XS GIS Cut Line= 2
2298861.87030742550101.751301912 2298963.0382656 550369.54883827
#Sta/Elev= 30
       0 2681.15    10.7 2674.06    13.8 2671.76      20 2666.46      25 2662.16
    29.3 2659.33    33.6 2657.13    37.9 2654.44    42.1 2652.55    50.7 2652.25
    60.3 2650.26    66.5 2649.68    80.6 2649.58    83.62649.629    89.2 2649.72
    93.5 2650.12   114.8 2653.53   119.1 2653.96   146.2 2653.58   156.5 2653.78
   174.7  2652.9   183.3 2651.95   187.6 2652.22   191.8 2653.56   204.6 2659.28
   215.5 2663.51   224.8 2666.61   247.4 2675.74   268.2 2685.94   286.3    2694
#Mann= 4 ,-1,0
       0     .06       0      20      .1       0    60.3    .045       0
    83.6      .1       0
Bank Sta=60.3,83.6
XS Rating Curve= 0 ,0
Exp/Cntr(USF)=0,0
Exp/Cntr=0.3,0.1

Type RM Length L Ch R = 1 ,1087    ,252.1,252.2,253.6
XS GIS Cut Line= 2
2298636.92037688550185.0660910012298752.37087033550442.151725906
#Sta/Elev= 30
       0  2680.4    14.7 2672.08    26.4 2666.02    44.9 2655.31    63.1 2649.09
    65.9 2648.15    70.3 2647.48    74.7 2647.76    81.2 2649.23    92.2 2650.98
     101  2650.2   109.7 2651.13   123.6 2651.78   138.7 2651.25   144.8 2650.75
   153.8 2648.77   159.9 2648.44   164.2  2648.7   171.1  2649.7   175.5 2650.85
   179.9 2652.37   184.1 2653.17   193.5  2653.7   196.2 2654.13   197.4  2654.5
   200.7 2656.52   206.2 2660.32   223.7 2669.25   250.1 2680.05   281.8 2693.86
#Mann= 3 ,-1,0
       0      .1       0    63.1    .045       0    81.2      .1       0
Bank Sta=63.1,81.2
XS Rating Curve= 0 ,0
Exp/Cntr(USF)=0,0
Exp/Cntr=0.3,0.1

Type RM Length L Ch R = 1 ,834     ,268.5,265.6,260.1
XS GIS Cut Line= 2
2298410.78023506550286.2340491812298545.27410888 550540.93926154
#Sta/Elev= 30
       0 2680.44    11.6 2674.82    21.4 2668.58      35 2660.56    44.7 2655.75
    51.6 2651.64    57.6 2649.18    80.1 2647.33    89.3  2644.8    98.3  2646.4
   102.8 2646.66   131.5 2645.74   143.6 2644.79   154.2 2644.92   161.6 2646.22
   165.7 2647.25     169 2647.57   184.3 2647.16   189.7 2647.83   202.4 2653.66
   206.9 2654.98   211.4 2655.74   216.4 2657.38   228.2 2664.46   238.5 2672.05
   242.8 2673.36   251.9 2675.22   265.7 2679.46   275.6  2683.9     288 2690.22
#Mann= 3 ,-1,0
       0      .1       0   131.5    .045       0   161.6      .1       0
Bank Sta=131.5,161.6
XS Rating Curve= 0 ,0
Exp/Cntr(USF)=0,0
Exp/Cntr=0.3,0.1
